--- STNKLKCK.prj (project) ---

Proj Title=STNKLKCK
Current Plan=p01
Default Exp/Contr=0,0
English Units
Geom File=g01
Flow File=f01
Plan File=p01
BEGIN DESCRIPTION:
END DESCRIPTION:
DSS Export Rating Curves= 0
DSS Export Rating Curve Sorted= 0
DSS Export Volume Flow Curves= 0
DXF Filename=..\STNKLKCK.
DXF OffsetX= 0
DXF OffsetY= 0
DXF ScaleX= 0
DXF ScaleY= 0

--- STNKLKCK.p01 (plan) ---

Plan Title=Floodplain
Program Version=4.00
Geom File=g01
Flow File=f01
K Sum by GR=0
Std Step Tol=0.01
Critical Tol=0.01
Num of Std Step Trials=20
Max Error Tol=0.3
Flow Tol Ratio=0.001
Split Flow NTrial=30
Split Flow Tol=0.02
Split Flow Ratio=0.02
Log Output Level=0
Friction Slope Method=1
Unsteady Friction Slope Method=2
Unsteady Bridges Friction Slope Method=1
Global Log Level=0
CheckData=False
Run HTab=0
Run UNet=0
Run PostProcess=0
UNET Theta=0
UNET Theta Warmup=0
UNET ZTol=0
UNET ZSATol=0
UNET MxIter=0
UNET MaxInSteps=0
UNET DtIC=0
UNET DtMin=0
UNET MaxCRTS=0
UNET WFStab=0
UNET SFStab=0
UNET WFX=0
UNET SFX=0
UNET DSS MLevel=0
UNET DZMax Abort=0
UNET Convert EG Bridges=0
UNET Use Existing IB Tables=0
UNET Froude Limit=0
UNET Froude Power=0
Write IC File=0
Echo Input=False
Echo Output=False
Write Detailed=0

--- STNKLKCK.f01 (steady flow) ---

Flow Title=NFF Regression Equation
Program Version=4.10
Number of Profiles= 1
Profile Names=P100yr
River Rch & RM=STNKLKCK,Main            ,13364.2
796.1914
River Rch & RM=STNKLKCK,Main            ,9201.9
 830.774
River Rch & RM=STNKLKCK,Main            ,8690.5
1019.196
River Rch & RM=STNKLKCK,Main            ,7540.7
1083.507
River Rch & RM=STNKLKCK,Main            ,4094.3
1165.019
Boundary for River Rch & Prof#=STNKLKCK,Main            , 1
Up Type= 0
Dn Type= 1
Dn Known WS=1606.9
DSS Import GetInterval= 0
DSS Import GetPeak= 0
DSS Import FillOption= 0

--- STNKLKCK.g01 (geometry) ---

Geom Title=USGS 10m DEM
Program Version=4.10

River Reach=STNKLKCK        ,Main
Reach XY= 30
     2023939.303       175222.31     2023771.298      175601.184
     2023878.243      175967.851     2023299.076      176210.212
     2023137.626      176663.515     2022776.854      176687.295
     2022468.326      176851.471      2022406.02      177019.934
     2022069.215      176894.239     2021604.785      177054.596
     2021636.035      177225.429     2021444.119      177409.132
      2021549.77      177822.712     2021007.833      178461.819
     2020510.187      179414.378     2020284.493      179474.101
     2020303.352      179927.838     2020103.243      180242.851
     2020113.659      180426.878      2020686.53      181186.143
     2020886.576      181707.434      2021140.06      181878.785
     2021208.104      182139.379     2021807.409      182597.017
     2022067.826      182411.601     2022219.909      182608.823
     2022210.882      183076.184     2022474.076      183235.212
     2022581.697      183573.304     2022912.303      183853.394

Type RM Length L Ch R = 1 ,13364.2 ,193,195.2,197.1
XS GIS Cut Line= 3
      2023705.48       175239.26     2024056.174      175256.622
     2024202.008      175135.094
#Sta/Elev= 30
       0 1761.86   20.661755.604    48.8 1748.44      65 1743.43    81.3 1737.84
   100.8 1732.05   113.8 1726.59   123.5 1723.21   133.3 1721.93   149.6 1721.35
  176.021721.493  193.09 1721.13   201.6 1719.78   211.3 1721.13   217.8 1721.77
   230.8 1722.14   240.6 1722.22   256.8 1721.56  341.061722.601  384.871723.296
   403.5 1723.62   429.7 1723.26     433 1723.12   439.5 1721.75   442.8 1721.51
   459.1 1723.83   462.4 1724.77   472.2 1729.05   521.3 1752.39     541  1760.3
#Mann= 7 ,-1 , 0
       0     .12       0   20.66     .06       0  176.02     .12       0
  193.09    .045       0   211.3     .06       0  341.06    .016       0
  384.87     .12       0
#XS Ineff= 2 , 0
                          310.23         1728.11
Permanent Ineff=
       F       F
Bank Sta=193.09,211.3
XS Rating Curve= 0 ,0
Exp/Cntr=0.3,0.1

Type RM Length L Ch R = 1 ,13168.9 ,208.5,206.3,202.9
XS GIS Cut Line= 2
     2023681.174      175414.608     2024164.826      175463.826
#Sta/Elev= 30
       0  1758.9    19.6 1754.15    52.2 1745.51    78.3 1737.06   104.4 1730.32
   114.2 1727.08   120.7 1725.63   130.5 1721.67   133.8  1721.1  158.671719.995
   189.2  1720.5   195.8 1720.03   202.3 1718.86   212.1 1720.12   215.3 1720.54
  222.231720.364   244.7 1720.21   257.8 1720.72   267.6 1720.24   316.5  1722.8
   332.8 1722.68   345.8 1723.42   362.2 1723.32   398.1 1724.23  417.051724.271
     447 1725.07  455.191725.618   466.6 1726.34   479.6 1726.38   486.2 1726.78
#Mann= 7 ,-1 , 0
       0     .06       0  158.67     .12       0   195.8    .045       0
   212.1     .12       0  222.23     .06       0  417.05    .016       0
  455.19     .06       0
Bank Sta=195.8,212.1
XS Rating Curve= 0 ,0
Exp/Cntr=0.3,0.1

Type RM Length L Ch R = 1 ,12962.6 ,198.2,203.1,203.7
XS GIS Cut Line= 4
     2023674.158      175551.066     2023732.751      175598.809
     2024072.378      175602.064     2024163.524      175650.892
#Sta/Elev= 30
       0 1743.69    15.8 1740.73    44.1 1734.57    69.3 1727.81    82.1 1723.86
   85.881723.266    95.2 1722.01   107.3 1719.26   111.5 1718.37     118  1717.8
   121.3 1718.29   124.6 1719.34  130.591719.945     216 1719.41   235.6 1719.73
   258.5 1719.34   268.3 1719.85   323.8 1719.97   392.4 1722.95   418.5 1723.12
  428.561724.398   457.2  1727.5   473.4 1731.83   476.6 1732.28   492.8 1732.09
  496.111732.398   499.2 1734.04   508.9 1741.02   512.2 1742.95   518.6 1745.14
#Mann= 7 ,-1 , 0
       0     .06       0   85.88     .12       0   107.3    .045       0
   124.6     .12       0  130.59     .06       0  428.56    .016       0
  496.11     .12       0
#XS Ineff= 2 , 0
                          325.57         1724.54
Permanent Ineff=
       F       F
Bank Sta=107.3,124.6
XS Rating Curve= 0 ,0
Exp/Cntr=0.3,0.1

Type RM Length L Ch R = 1 ,12759.6 ,375.1,394.2,409.4
XS GIS Cut Line= 4
      2023550.46      175708.401     2023608.836      175755.493
     2024054.149      175754.191     2024142.908      175810.615
#Sta/Elev= 30
       0 1742.92    16.3 1733.02    26.1 1728.36   29.391727.333    39.1 1724.78
    52.2 1722.84      62 1722.13     111 1721.49   143.8 1721.74   153.6 1721.44
     170 1719.29   179.8 1718.63   274.7 1719.14   287.8 1718.54   294.4 1717.52
   304.2 1718.45     314  1718.9   389.3 1719.18  442.921718.604   500.7  1719.9
     517 1723.03  525.621727.136   539.4  1733.9     549 1741.14  574.151743.767
   580.9 1744.75   584.1 1746.54   593.6 1754.88   596.8 1756.98   625.5    1770
#Mann= 7 ,-1 , 0
       0     .12       0   29.39     .06       0   287.8    .045       0
   304.2     .06       0  442.92     .12       0  525.62    .016       0
  574.15     .12       0
#XS Ineff= 2 , 0
          182.95 1724.52  461.36         1725.75
Permanent Ineff=
       F       F
Bank Sta=287.8,304.2
XS Rating Curve= 0 ,0
Exp/Cntr=0.3,0.1

Type RM Length L Ch R = 1 ,12365.4 ,387.9,385.1,378.1
XS GIS Cut Line= 2
     2023541.851      175755.754     2023934.213      176155.059
#Sta/Elev= 30
       0 1733.84    22.9 1725.62   28.131724.417    39.3 1722.47    55.6 1721.81
   114.6 1720.91   124.4 1721.24   209.5 1720.45     275 1718.08   291.4 1716.63
   333.9 1717.69   353.6 1717.17  369.991716.007     374 1715.46     383  1714.4
   386.3 1714.57   389.6 1715.42   392.8 1717.99   399.4 1726.37   402.7 1729.29
     406 1730.36   409.2 1730.67   422.3 1730.63   425.6 1731.84  436.611740.228
     442 1742.84   491.1 1759.96     514 1767.39   540.2  1774.7   559.8 1779.12
#Mann= 6 ,-1 , 0
       0     .12       0   28.13     .06       0  369.99     .12       0
     374    .045       0   389.6    .016       0  436.61     .12       0
Bank Sta=374,389.6
XS Rating Curve= 0 ,0
Exp/Cntr=0.3,0.1

Type RM Length L Ch R = 1 ,11980.3 ,198.2,205.4,212.8
XS GIS Cut Line= 2
     2023343.501      176032.229     2023619.542      176313.479
#Sta/Elev= 30
       0 1767.29    29.3 1743.79    42.3 1735.01   49.781730.449    65.1 1722.03
    71.6  1719.4    74.9 1718.75   107.5 1717.49   117.2 1715.84   156.3 1714.58
   172.6 1713.45   185.6 1712.85   192.9 1713.47  211.831714.769  221.231715.532
   276.8 1718.95   293.1 1721.28  314.911723.007   319.2 1723.83   322.4 1725.33
   325.7 1725.94     342 1725.61   345.2 1725.97   348.5 1728.36  349.291729.276
   351.7 1732.07     355 1735.05   358.3 1736.48   377.8 1743.58   394.1 1748.34
#Mann= 8 ,-1 , 0
       0     .12       0   49.78     .06       0   172.6    .045       0
   192.9     .06       0  211.83     .12       0  221.23     .06       0
  314.91    .016       0  349.29     .12       0
Bank Sta=172.6,192.9
XS Rating Curve= 0 ,0
Exp/Cntr=0.3,0.1

Type RM Length L Ch R = 1 ,11774.9 ,339.5,328.5,315.9
XS GIS Cut Line= 2
     2023188.119      176115.997     2023514.508      176470.163
#Sta/Elev= 30
       0 1805.52     9.8 1797.98    19.7 1788.17    22.9 1786.54    29.5 1784.77
    32.8 1782.89    39.3 1776.85    68.8 1755.85    85.2 1743.52    98.3 1732.62
   104.8 1728.24   121.2 1718.57   127.8 1716.23   139.5 1713.26   144.2 1711.98
   157.3 1713.03   183.5 1714.53   245.7 1714.45   278.5 1715.15   291.6 1716.71
   327.6    1718   347.3 1720.48  356.881722.468   370.2 1725.33   383.3 1731.64
   396.4    1732   399.7 1732.94  410.521739.046   458.7 1755.34   481.6 1762.31
#Mann= 5 ,-1 , 0
       0     .12       0   139.5    .045       0   157.3     .06       0
  356.88    .016       0  410.52     .12       0
#XS Ineff= 2 , 0
                          256.39         1724.46
Permanent Ineff=
       F       F
Bank Sta=139.5,157.3
XS Rating Curve= 0 ,0
Exp/Cntr=0.3,0.1

Type RM Length L Ch R = 1 ,11446.5 ,384.7,405.1,421.4
XS GIS Cut Line= 3
     2022976.313      176359.052     2023070.063      176487.524
     2023422.494      176593.427
#Sta/Elev= 30
       0 1765.77      26 1756.29    58.4 1743.04    81.1 1735.73    97.4 1731.28
   113.6 1727.82   149.3 1721.74     159 1720.23   188.4 1717.66  214.541712.505
   227.4 1710.72   240.5 1710.17     247 1710.66     260 1712.37   279.5  1712.8
   321.9 1715.48   338.2 1718.33  351.651723.007     361 1725.59  388.371729.467
     400 1732.43   419.6 1732.04   422.8 1732.66   429.3 1735.38  433.991736.015
   452.1 1735.74   478.2 1740.92     488 1743.93   517.3  1755.6     527 1758.58
#Mann= 7 ,-1 , 0
       0     .12       0  214.54     .06       0   227.4    .045       0
     247     .06       0  351.65     .12       0  388.37    .016       0
  433.99     .12       0
Bank Sta=227.4,247
XS Rating Curve= 0 ,0
Exp/Cntr=0.3,0.1

Type RM Length L Ch R = 1 ,11041.4 ,235.6,236.5,235.2
XS GIS Cut Line= 2
     2022847.557      176529.127     2023015.086      176881.795
#Sta/Elev= 30
       0 1738.67     9.8 1734.83    29.3 1728.62      39 1725.97   65.111720.038
    78.1 1717.66   104.1 1714.93   120.4 1712.43   130.2 1711.51   156.2 1711.22
   167.3 1708.77   175.7 1708.08   182.3 1709.02  183.971709.276     192 1710.07
   211.5 1710.56  250.241709.175   253.8 1709.65     257 1711.67   260.3  1712.9
   266.8 1713.45   279.8 1713.52   283.1 1714.45  284.851716.145   289.6 1720.43
   292.8 1722.63   318.9 1737.65   338.4  1750.1   361.2 1762.58   390.4 1777.43
#Mann= 7 ,-1 , 0
       0     .12       0   65.11     .06       0   167.3    .045       0
   182.3     .06       0  183.97     .12       0  250.24    .016       0
  284.85     .12       0
#XS Ineff= 2 , 0
                          243.18         1720.38
Permanent Ineff=
       F       F
Bank Sta=167.3,182.3
XS Rating Curve= 0 ,0
Exp/Cntr=0.3,0.1

Type RM Length L Ch R = 1 ,10804.9 ,330.2,324.1,318.7
XS GIS Cut Line= 2
     2022649.924      176584.747     2022804.149       176928.67
#Sta/Elev= 30
       0 1749.07    16.4 1743.78    42.6 1736.75    72.1 1729.81    81.9 1725.56
    88.5 1723.47      95 1720.71  111.291715.003     118 1712.68  123.861711.697
   134.4 1710.66   147.5  1708.4     162 1707.45   173.7 1706.56   180.3 1707.25
   193.4 1707.83   206.5 1710.45  214.64 1711.13   226.2 1710.35   229.4 1711.79
   232.7 1713.83     236 1714.92     2491716.876   268.8 1719.96   285.2 1723.08
   311.4 1730.08   327.8 1735.52   334.3 1738.25   350.7 1744.18   376.9 1755.47
#Mann= 7 ,-1 , 0
       0     .12       0  111.29     .06       0  123.86     .12       0
     162    .045       0   180.3     .12       0  214.64    .016       0
     249     .12       0
Bank Sta=162,180.3
XS Rating Curve= 0 ,0
Exp/Cntr=0.3,0.1

Type RM Length L Ch R = 1 ,10480.8 ,354.6,383.3,407.5
XS GIS Cut Line= 3
     2022387.482      176724.243     2022396.597       176834.92
     2022568.472      177035.441
#Sta/Elev= 30
       0 1727.98     6.5 1726.34    29.4 1721.66    68.6 1715.86   107.8 1711.07
   117.6 1710.69  134.481709.321   143.7  1709.3   146.9 1708.64   156.7 1705.94
   166.5 1702.67   176.3 1702.25   184.1 1702.96   189.3 1703.68   195.8 1703.18
   202.4  1703.9   212.1 1704.26   228.4 1703.27  255.691706.386     261 1707.18
   270.8 1710.31   274.1 1710.69   287.1 1710.59   290.4 1711.19  297.361714.448
   306.7 1718.04     323 1725.22   352.3 1741.02   362.1 1745.87   375.2 1753.38
#Mann= 6 ,-1 , 0
       0     .06       0  134.48     .12       0   166.5    .045       0
   184.1     .12       0  255.69    .016       0  297.36     .12       0
Bank Sta=166.5,184.1
XS Rating Curve= 0 ,0
Exp/Cntr=0.3,0.1

Type RM Length L Ch R = 1 ,10097.4 ,231.4,215.1,197.9
XS GIS Cut Line= 4
     2022246.857      176721.639     2022236.441      176817.993
     2022148.188      177029.191     2022177.702      177173.288
#Sta/Elev= 30
       0 1730.51    19.4 1726.81    29.1 1724.14    45.2 1721.03    67.8 1715.77
    80.8 1713.16   88.251712.169  103.141709.561   149.2 1701.97     1611701.508
     195 1701.16   221.2 1698.01   234.2 1697.53     239 1697.88   263.7 1698.45
     280 1699.88   289.8 1701.57     316 1707.26   325.8 1710.05   342.2 1715.76
   355.2 1721.67  382.84 1731.81   391.2 1735.44   394.4 1736.13   407.5 1736.26
   410.8 1736.84   417.3 1741.19   420.6 1742.81  433.93 1746.63   472.9 1756.59
#Mann= 8 ,-1 , 0
       0     .12       0   88.25     .06       0  103.14     .12       0
     161     .06       0   221.2    .045       0     239     .12       0
  382.84    .016       0  433.93     .12       0
Bank Sta=221.2,239
XS Rating Curve= 0 ,0
Exp/Cntr=0.3,0.1

Type RM Length L Ch R = 1 ,9882.3  ,319.6,319.9,319.5
XS GIS Cut Line= 3
     2021950.272      176657.663     2021929.438      176763.566
     2022078.744      177178.497
#Sta/Elev= 30
       0 1772.98    22.9 1752.66    55.6 1725.95      85 1707.47    91.6 1702.58
    94.8 1701.12   107.9 1697.74   114.5  1697.2  196.541696.675  201.131696.673
   254.9 1698.12   265.2 1693.98   274.5 1692.02   284.3 1692.99   294.1 1693.61
   310.4 1692.89   320.2  1694.6   346.4  1696.6  376.93  1697.2  392.49  1697.3
   405.2    1698     415 1700.48   431.3 1706.89   460.7 1721.68   480.3 1728.89
  505.881735.829     513 1738.61   529.3 1738.69     5391741.092   548.9 1743.24
#Mann= 9 ,-1 , 0
       0     .12       0  196.54     .06       0  201.13     .12       0
   265.2    .045       0   284.3     .12       0  376.93     .06       0
  392.49     .12       0  505.88    .016       0     539     .12       0
Bank Sta=265.2,284.3
XS Rating Curve= 0 ,0
Exp/Cntr=0.3,0.1

Type RM Length L Ch R = 1 ,9562.4  ,381.7,360.6,334.5
XS GIS Cut Line= 4
     2021622.291      176750.719     2021634.444      176879.191
     2021740.347       177172.16      2021886.18      177229.451
#Sta/Elev= 30
       0  1722.4      29  1707.1    38.7 1702.62    48.4 1697.45    51.6 1696.65
    58.1 1696.03    64.5  1694.6    77.4  1693.6   106.5 1693.22   138.9 1691.78
   214.3 1689.87     234 1689.92   240.5 1689.53   248.3 1687.84   256.9 1686.41
   260.2 1686.82   263.3 1687.97     270 1689.26   283.2 1690.05  321.041689.978
   368.4 1689.78   381.5 1690.38   397.9 1692.29   411.1 1693.33   450.4 1693.36
   479.7 1694.73   496.1 1696.18   522.2 1700.13   551.6 1703.69   597.2 1711.32
#Mann= 4 ,-1 , 0
       0     .12       0   248.3    .045       0   263.3     .12       0
  321.04     .06       0
#XS Ineff= 2 , 0
          190.91 1694.78
Permanent Ineff=
       F       F
Bank Sta=248.3,263.3
XS Rating Curve= 0 ,0
Exp/Cntr=0.3,0.1

Type RM Length L Ch R = 1 ,9201.9  ,521.7,511.3,499.2
XS GIS Cut Line= 3
     2021270.295      177252.889     2021420.758      177228.844
      2021854.93      177336.222
#Sta/Elev= 30
       0 1759.38    35.7 1747.29      94 1722.11   132.9 1707.36  143.451704.003
   152.4 1700.13   162.2 1694.35   168.7 1692.14   181.8 1690.48  210.851688.882
   220.9 1689.24   253.6 1688.85   266.6 1687.41     283 1687.69     296 1686.07
   315.6 1685.54  319.78  1686.1   325.4 1687.95   328.7 1688.48  347.511688.205
   367.8 1687.64   377.6 1688.12   387.4 1689.63   403.8 1690.87   472.3 1692.62
   488.6 1693.96   514.8 1694.74   553.9 1700.46   583.3 1706.37   599.6 1710.42
#Mann= 6 ,-1 , 0
       0     .12       0  143.45     .06       0  210.85     .12       0
     296    .045       0  319.78     .12       0  347.51     .06       0
Bank Sta=296,319.78
XS Rating Curve= 0 ,0
Exp/Cntr=0.3,0.1

Type RM Length L Ch R = 1 ,8690.5  ,397.9,403.6,414.3
XS GIS Cut Line= 4
     2021241.649      177668.254     2021409.618      177702.108
     2021668.732       177647.42     2021832.795      177676.066
#Sta/Elev= 30
       0 1753.79    25.9 1740.23      42 1733.05    67.9  1722.6    77.6 1720.33
   126.1 1704.96  145.291699.849   161.6 1695.34  190.251691.081   210.6 1688.68
   236.7 1687.37  248.52 1684.76   256.4 1683.02   262.9 1683.74   264.9 1684.63
   269.4 1686.16  273.441686.491   387.1 1686.66  411.791687.697   439.4 1691.43
   468.8 1697.92  476.63 1700.46   481.9 1702.31   498.2 1702.39   501.5  1702.9
  507.621706.711   511.3  1708.3   534.1 1715.12   592.9 1736.28   602.7 1739.15
#Mann= 9 ,-1 , 0
       0     .12       0  145.29     .06       0  190.25     .12       0
  248.52    .045       0   264.9     .12       0  273.44     .06       0
  411.79     .12       0  476.63    .016       0  507.62     .12       0
Bank Sta=248.52,264.9
XS Rating Curve= 0 ,0
Exp/Cntr=0.3,0.1

Type RM Length L Ch R = 1 ,8286.9  ,315.6,330.5,344.5
XS GIS Cut Line= 2
      2021205.11      177896.261      2021728.42      178024.968
#Sta/Elev= 30
       0 1723.51    6.871721.889    39.2 1715.79    75.1 1707.11   101.2 1700.12
  137.861692.552   156.8 1689.69   166.6 1685.35  175.65 1683.33   179.6 1682.22
   194.7 1683.33   202.5  1685.1   215.6 1685.43  228.381684.875   235.2 1686.37
   241.7 1686.96   297.2 1686.07   313.5 1686.56   369.1 1686.52   385.4 1687.66
  398.531689.945   424.6 1696.11  460.481705.655     467 1708.48   470.3 1709.08
   486.6 1709.64   489.9 1711.49  493.051714.105   496.4 1716.45   538.9 1731.21
#Mann= 9 ,-1 , 0
       0     .12       0    6.87     .06       0  137.86     .12       0
  175.65    .045       0   194.7     .12       0  228.38     .06       0
  398.53     .12       0  460.48    .016       0  493.05     .12       0
#XS Ineff= 2 , 0
                          348.58         1692.69
Permanent Ineff=
       F       F
Bank Sta=175.65,194.7
XS Rating Curve= 0 ,0
Exp/Cntr=0.3,0.1

Type RM Length L Ch R = 1 ,7956.4  ,424.1,415.7,406.1
XS GIS Cut Line= 2
       2021130.8      178051.542     2021434.674      178426.979
#Sta/Elev= 30
       0 1719.21     6.5 1717.47    19.6  1714.9    32.6  1711.5      62 1705.84
    84.8 1700.35    94.6 1698.78     111  1695.5   130.5    1693   140.3 1691.24
   146.9 1690.46   169.7 1684.11   176.2 1683.54   195.8 1684.02   205.6 1683.21
   215.3 1681.69   228.4 1680.88   231.7 1680.98     235 1682.03   241.5 1684.57
   244.8 1685.38   254.6 1686.42   283.9 1686.11   368.8 1689.26   385.1 1690.45
   414.5 1690.96   430.8 1692.21   453.6 1692.05     470  1693.1     483 1694.67
#Mann= 3 ,-1 , 0
       0     .12       0   215.3    .045       0     235     .12       0
Bank Sta=215.3,235
XS Rating Curve= 0 ,0
Exp/Cntr=0.3,0.1

Type RM Length L Ch R = 1 ,7540.7  ,331.8,337,339.4
XS GIS Cut Line= 3
     2020788.883      178471.463     2020919.901      178481.034
     2021259.519      178660.617
#Sta/Elev= 30
       0 1755.26    28.8 1738.81    64.1 1717.85    80.1  1709.9    92.9 1704.63
   121.8  1695.7   141.1 1691.88   170.4 1682.67   180.2 1680.61   196.5 1680.54
   199.7 1680.22     203 1679.18   209.5 1677.52   214.4 1677.36   219.3 1677.69
   222.5 1679.68   225.8 1681.02     229 1681.28   264.8 1681.13   281.1 1682.95
   333.2 1683.84   346.2 1684.78   359.3 1687.44   372.3 1690.96   385.3 1695.21
   398.3 1698.55   460.2 1703.59  503.461708.973   512.3 1710.23   515.5 1711.68
#Mann= 4 ,-1 , 0
       0     .12       0     203    .045       0   222.5     .12       0
  503.46    .016       0
Bank Sta=203,222.5
XS Rating Curve= 0 ,0
Exp/Cntr=0.3,0.1

Type RM Length L Ch R = 1 ,7203.7  ,207.6,207.5,207.5
XS GIS Cut Line= 3
     2020707.361      178738.566     2020827.845      178782.107
      2021083.58      178978.993
#Sta/Elev= 30
       0 1795.67     6.4 1792.17    19.2 1783.81    57.6 1753.97    67.3  1745.2
    70.5 1743.05    80.1 1738.28    99.3 1722.26   128.1 1701.76   147.7 1689.19
   157.4 1683.63     164 1681.56   180.3 1679.76     195 1677.18   199.8 1676.61
   209.6 1676.71  210.97 1677.22   216.1 1679.58   219.4 1680.23   232.4 1679.97
     265 1680.81   281.3 1681.76   300.9  1683.7     327 1689.03  364.631697.926
   375.9 1702.54   395.4 1703.11  405.291705.434   424.8 1710.75   450.9 1719.99
#Mann= 5 ,-1 , 0
       0     .12       0     195    .045       0  210.97     .12       0
  364.63    .016       0  405.29     .12       0
Bank Sta=195,210.97
XS Rating Curve= 0 ,0
Exp/Cntr=0.3,0.1

Type RM Length L Ch R = 1 ,6996.2  ,236.5,235.3,232.3
XS GIS Cut Line= 2
     2020629.636      178888.671     2020939.599      179129.259
#Sta/Elev= 30
       0 1767.02    26.2 1750.54    32.7 1746.02    68.7  1717.9    94.8 1696.38
   104.6 1689.15   111.2 1683.63   114.4 1681.81     121 1680.26   134.1 1679.34
   150.4 1678.68   166.8 1679.32     170 1679.08   173.3 1678.13   176.6 1676.73
   179.8 1676.06   186.4  1676.5   189.6 1677.45   202.7 1680.14   232.2 1682.59
   264.8 1687.14   317.2 1696.86  330.35 1697.21   346.6 1699.81   359.7    1700
     363 1700.73   366.2 1702.68   369.5 1703.99   385.8 1705.43   392.4 1706.54
#Mann= 4 ,-1 , 0
       0     .12       0   173.3    .045       0   189.6     .12       0
  330.35    .016       0
Bank Sta=173.3,189.6
XS Rating Curve= 0 ,0
Exp/Cntr=0.3,0.1

Type RM Length L Ch R = 1 ,6760.8  ,138.6,136,134.5
XS GIS Cut Line= 3
     2020524.201      179077.108      2020535.92       179120.51
      2020817.17      179304.972
#Sta/Elev= 30
       0 1703.27     6.4 1701.09    16.1 1699.28      45 1691.32    54.8 1689.31
    90.7  1684.9   103.7  1682.2   110.3 1681.28   120.1 1678.29   133.1 1677.66
   137.7 1676.56   146.2 1675.88   152.7 1676.51   159.2  1678.3  162.341678.576
     218 1679.29   227.8  1679.9     254 1682.07   270.3 1684.04   276.8  1685.2
  288.85 1688.33   306.2 1694.23   319.3 1695.61   325.8 1699.03   342.1 1699.74
   351.9 1705.77  356.021707.678   361.7 1709.63     365 1710.05   381.3 1710.42
#Mann= 6 ,-1 , 0
       0     .12       0   137.7    .045       0   152.7     .12       0
  162.34     .06       0  288.85    .016       0  356.02     .12       0
Bank Sta=137.7,152.7
XS Rating Curve= 0 ,0
Exp/Cntr=0.3,0.1

Type RM Length L Ch R = 1 ,6624.8  ,58.1,58.8,59.2
XS GIS Cut Line= 3
     2020476.892      179167.385     2020515.086      179269.816
     2020788.524      179410.441
#Sta/Elev= 30
       0 1696.82    16.1 1694.94    51.4 1689.45    61.1 1685.76      74 1683.44
    83.6 1682.62   102.9 1682.68   119.1 1681.72   122.4 1680.83     129 1677.48
   134.4 1676.49   145.3 1675.86  150.58 1676.51   158.4 1678.25  191.441677.341
   204.2 1676.51     214 1676.78   233.6 1678.51  263.661682.557   279.4    1684
     299  1690.6   305.6 1693.34   312.1 1697.33  316.281700.596   318.7 1701.85
   321.9 1702.32   331.8 1702.78  349.061710.352   390.6 1723.39   416.8 1730.12
#Mann= 7 ,-1 , 0
       0     .12       0   134.4    .045       0  150.58     .12       0
  191.44     .06       0  263.66     .12       0  316.28    .016       0
  349.06     .12       0
#XS Ineff= 2 , 0
          123.58 1682.66
Permanent Ineff=
       F       F
Bank Sta=134.4,150.58
XS Rating Curve= 0 ,0
Exp/Cntr=0.3,0.1

Type RM Length L Ch R = 1 ,6566.1  ,95.2,112,128.1
XS GIS Cut Line= 2
     2020364.045      179255.927     2020765.086      179462.524
#Sta/Elev= 30
       0 1700.83   18.91 1694.42    26.2 1691.63    39.2 1690.81    55.6 1686.13
    65.4 1684.06  122.431681.615   163.4 1679.54     170  1678.3   176.5 1675.79
   186.3 1674.98   193.3 1676.13   202.7 1677.53   225.6 1676.41   261.5 1676.94
   274.6 1678.49  280.741680.143   300.8 1687.06  307.971688.435  312.121689.011
   317.1 1690.86     340 1702.36   356.3 1703.13   362.9 1706.99  370.091708.785
   382.5 1712.08   408.6 1720.62   421.7 1723.39   441.3 1725.83   451.1 1729.57
#Mann= 9 ,-1 , 0
       0     .12       0   18.91     .06       0  122.43     .12       0
   176.5    .045       0   193.3     .12       0  280.74     .06       0
  307.97     .12       0  312.12    .016       0  370.09     .12       0
Bank Sta=176.5,193.3
XS Rating Curve= 0 ,0
Exp/Cntr=0.3,0.1

Type RM Length L Ch R = 1 ,6454.1  ,130.8,134.3,138
XS GIS Cut Line= 4
     2020334.893      179270.265     2020446.872      179336.237
      2020510.24      179502.035     2020601.386      179561.063
#Sta/Elev= 30
       0 1706.85    19.5 1698.49    35.7  1693.1    48.7 1690.15    58.5 1687.25
    71.5 1686.06    87.7 1682.91   110.5 1680.76   162.2 1677.72   178.4 1676.96
   207.4 1676.63   220.3 1675.67   236.5 1674.16   249.4 1672.86   255.8 1673.02
   262.3 1674.37     272 1677.52   281.6 1683.54   288.1 1685.91   307.5 1685.94
   320.2 1687.59   345.8 1689.76   355.4 1691.83   371.3 1698.09   377.7 1699.54
   393.7 1699.44   396.9 1700.47   403.3 1704.43   412.9 1706.59     416 1707.52
#Mann= 7 ,-1 , 0
       0     .12       0    87.7     .06       0   220.3     .12       0
   236.5    .045       0   262.3     .12       0   371.3    .016       0
   412.9     .12       0
Bank Sta=236.5,262.3
XS Rating Curve= 0 ,0
Exp/Cntr=0.3,0.1

Type RM Length L Ch R = 1 ,6319.8  ,297.4,276.3,255.4
XS GIS Cut Line= 4
     2020283.316      179350.545     2020343.211      179384.399
     2020378.368      179566.691     2020518.993      179646.118
#Sta/Elev= 30
       0 1707.89     9.8 1702.13    22.9 1695.91    29.5 1691.75    32.8 1690.24
    42.6 1688.32    52.4 1684.95    62.2 1682.46    85.1 1678.36    98.1 1675.14
  121.151672.602   130.7 1671.58   140.5 1670.89     147 1671.99   150.7  1672.7
   163.3 1674.31   176.3 1677.83  193.791678.354   251.2 1680.18  313.671684.184
  338.571685.285     361    1687   367.5 1688.71   377.2 1692.17  381.521692.527
   386.9 1692.69   390.1 1693.32   399.8 1698.44   412.7  1699.4     416 1700.81
#Mann= 9 ,-1 , 0
       0     .12       0  121.15     .06       0   130.7    .045       0
     147     .06       0   150.7     .12       0  193.79     .06       0
  313.67     .08       0  338.57     .06       0  381.52    .016       0
Bank Sta=130.7,147
XS Rating Curve= 0 ,0
Exp/Cntr=0.3,0.1

Type RM Length L Ch R = 1 ,6043.5  ,305,307.1,306.4
XS GIS Cut Line= 2
     2020063.698      179578.844     2020438.698      179761.135
#Sta/Elev= 30
       0 1727.02    32.6 1710.95    39.1 1707.25    48.9 1701.02    68.4 1686.34
    74.9 1682.16    81.4 1678.49      88 1675.97    97.7 1674.68   107.5 1674.25
   182.4 1674.32   192.1 1671.84   198.7 1669.59   208.5 1668.51     215 1669.54
   218.2 1671.63   221.5 1673.66     228 1675.93     2461677.383   299.7  1677.7
  340.641679.307   361.6 1680.08   371.4 1681.57   377.9 1683.19  392.571690.316
   400.7 1695.09   403.9  1696.3   410.4 1696.68   413.7 1697.72     417 1699.71
#Mann= 6 ,-1 , 0
       0     .12       0   192.1    .045       0   218.2     .12       0
     246     .06       0  340.64     .12       0  392.57    .016       0
#XS Ineff= 2 , 0
          120.74  1682.2
Permanent Ineff=
       F       F
Bank Sta=192.1,218.2
XS Rating Curve= 0 ,0
Exp/Cntr=0.3,0.1

Type RM Length L Ch R = 1 ,5736.4  ,161.5,160.9,159.3
XS GIS Cut Line= 3
     2019997.291      179844.469      2020080.65      179844.652
     2020456.059      180009.399
#Sta/Elev= 30
       0 1691.84      16 1689.57    32.1 1685.12    44.9 1682.85    86.6 1679.95
    99.8 1678.32   112.9 1679.03   135.8 1678.82   175.2 1675.82   214.6 1675.94
   224.4 1674.74   283.4 1671.77   309.7 1671.67   316.2  1670.1   322.8 1667.66
   329.3  1668.1  334.07 1669.99   335.9 1671.37   345.7 1685.34     349 1687.79
   352.3 1688.83   362.1 1690.12   365.4 1692.64  369.861697.736   375.3 1702.58
   378.5 1704.38   427.7 1730.06   440.8 1735.65   476.9 1748.56   493.3 1752.35
#Mann= 4 ,-1 , 0
       0     .12       0   316.2    .045       0  334.07    .016       0
  369.86     .12       0
Bank Sta=316.2,334.07
XS Rating Curve= 0 ,0
Exp/Cntr=0.3,0.1

Type RM Length L Ch R = 1 ,5575.5  ,134.8,133.6,131.9
XS GIS Cut Line= 3
     2019961.701      179974.243       2020232.1      180077.108
      2020410.92      180070.163
#Sta/Elev= 30
       0 1687.02    55.3  1687.1    68.3 1688.16    71.5 1687.88    87.8 1684.36
     104 1682.26   120.3 1681.22   149.5 1676.49     169 1675.07   237.3 1671.87
   250.3 1670.07   253.4 1669.17     260 1666.91   266.6 1667.26     273 1668.99
  280.411670.818   282.8 1671.55   289.3 1675.15   292.6 1675.69   305.6 1675.98
   308.8 1677.16   315.3 1681.78  328.641688.669   364.1 1706.32   390.2 1715.58
   403.2 1721.08   422.7 1726.74   432.5 1729.03   442.2 1732.33   468.3 1739.57
#Mann= 5 ,-1 , 0
       0     .12       0   253.4    .045       0     273     .12       0
  280.41    .016       0  328.64     .12       0
Bank Sta=253.4,273
XS Rating Curve= 0 ,0
Exp/Cntr=0.3,0.1

Type RM Length L Ch R = 1 ,5441.9  ,158,140,121.2
XS GIS Cut Line= 3
     2019925.243      180103.149     2020242.951      180217.733
     2020366.649      180190.389
#Sta/Elev= 30
       0 1699.79    75.4 1691.25    98.4 1689.48   108.2 1687.92   114.8  1686.3
   124.6 1682.18     141 1673.62   147.6    1672   203.3 1671.31   213.1 1670.48
     221  1668.5   229.5 1666.87   232.8 1666.82     236 1666.98   239.4 1667.93
  240.06 1668.79   245.9 1671.18   249.2 1671.76   262.3 1671.67  272.491673.928
   278.7 1674.73   301.7 1674.93   318.1 1677.24   334.5 1678.73   350.7 1681.49
  363.641687.808   396.2 1701.47   448.2 1713.83   454.7 1715.79   464.4 1719.62
#Mann= 5 ,-1 , 0
       0     .12       0     221    .045       0  240.06     .12       0
  272.49    .016       0  363.64     .12       0
Bank Sta=221,240.06
XS Rating Curve= 0 ,0
Exp/Cntr=0.3,0.1

Type RM Length L Ch R = 1 ,5301.9  ,148.3,128.6,73.5
XS GIS Cut Line= 3
     2019896.597       180424.33     2020224.722      180242.038
     2020339.305      180228.149
#Sta/Elev= 30
       0 1737.95    13.1 1733.08    22.8 1728.53    35.9 1724.31    88.1 1703.26
   107.7 1696.37   159.9 1680.06     173 1673.71   179.5  1671.3     186 1670.21
   202.4  1670.6   218.7 1670.18     222 1669.42   225.2 1667.84   228.5 1666.66
   238.3 1666.37   244.9 1667.38   251.3 1669.92   261.1 1671.62   274.2 1672.61
  305.051673.056   339.5 1673.51  352.871675.304  387.891678.882   391.4 1679.47
   404.2 1683.36   413.8 1684.51   424.81688.879   455.5 1699.79   490.8 1709.73
#Mann= 7 ,-1 , 0
       0     .12       0   225.2    .045       0   244.9     .12       0
  305.05    .016       0  352.87     .12       0  387.89    .016       0
   424.8     .12       0
Bank Sta=225.2,244.9
XS Rating Curve= 0 ,0
Exp/Cntr=0.3,0.1

Type RM Length L Ch R = 1 ,5173.3  ,47.3,45,78.8
XS GIS Cut Line= 4
     2019993.385      180537.177      2020102.76      180493.774
     2020146.597      180336.222     2020370.555      180269.816
#Sta/Elev= 30
       0 1727.02    29.4 1715.91    65.4 1702.95   101.3 1688.11   111.1  1684.5
   117.7 1680.66   137.3 1673.33   143.8  1671.8   163.5 1670.14   172.3 1667.67
   176.6  1666.6   183.1 1666.18   186.4 1666.31   192.9 1667.45     206 1670.08
   212.5 1670.77   258.3 1671.97  284.45 1672.13   300.7 1671.68     325 1672.25
   346.1 1673.02   355.8 1673.85   378.5 1677.36   401.2 1681.82  414.471685.092
   427.2 1688.95   436.9 1690.38  454.911697.268   508.3  1711.8   514.8 1714.09
#Mann= 7 ,-1 , 0
       0     .12       0   172.3    .045       0   192.9     .12       0
  284.45    .016       0     325     .12       0  414.47    .016       0
  454.91     .12       0
Bank Sta=172.3,192.9
XS Rating Curve= 0 ,0
Exp/Cntr=0.3,0.1

Type RM Length L Ch R = 1 ,5128.3  ,83.5,107.1,129.3
XS GIS Cut Line= 4
     2020026.371      180559.747     2020135.746      180516.344
     2020175.243      180360.962     2020387.482      180289.347
#Sta/Elev= 30
       0 1717.39      36 1704.84   83.551685.741      85 1684.99    91.5 1679.09
    94.8 1677.11   117.7 1675.62   153.7 1669.18   159.2 1667.34   163.5  1666.3
   166.8 1666.18   176.6 1666.25   179.8 1666.82   189.6 1670.28   202.7 1670.71
   215.8 1671.87   258.4 1671.27  283.361671.786   320.2 1671.96   339.7 1673.86
   378.6 1680.15  398.731684.932   411.1 1689.73   420.8 1691.39   424.1 1692.46
   430.6  1695.4  441.41 1699.33     463 1705.86   479.3 1710.12     502 1718.47
#Mann= 7 ,-1 , 0
       0     .12       0   83.55    .016       0   159.2    .045       0
   179.8    .016       0  283.36     .12       0  398.73    .016       0
  441.41     .12       0
Bank Sta=159.2,179.8
XS Rating Curve= 0 ,0
Exp/Cntr=0.3,0.1

Type RM Length L Ch R = 1 ,5021.2  ,249.5,247.5,241.9
XS GIS Cut Line= 3
     2020033.316      180598.809      2020138.35      180590.997
     2020412.656      180460.788
#Sta/Elev= 30
       0 1716.38    19.2  1710.5   58.931697.247    63.8  1695.3    73.4 1687.37
    76.6 1685.52    79.8 1684.92    89.4 1684.89   94.271684.197   102.1 1680.83
   118.4 1677.68     138 1672.72   144.5 1671.66   160.8 1670.47   167.4 1668.84
   171.6 1666.99   173.9 1666.36   180.4 1666.22   186.6 1666.77   193.5 1669.33
   196.7 1669.91   226.1 1669.76   235.9    1671   281.6 1673.92   304.5 1676.92
   330.6 1682.49   350.2 1688.26  390.01 1697.38   399.2 1701.04     409 1701.89
#Mann= 6 ,-1 , 0
       0     .12       0   58.93    .016       0   94.27     .12       0
   171.6    .045       0   186.6     .12       0  390.01    .016       0
Bank Sta=171.6,186.6
XS Rating Curve= 0 ,0
Exp/Cntr=0.3,0.1

Type RM Length L Ch R = 1 ,4773.7  ,369.8,371.8,368.7
XS GIS Cut Line= 2
     2020159.184      180847.073     2020493.385      180606.622
#Sta/Elev= 30
       0 1699.99    35.9 1690.86    52.3 1685.88   59.161682.973   66.721679.764
    68.6    1679    75.2 1678.05    94.8 1677.57   114.4 1676.31   127.4 1676.17
     134  1675.7   150.3 1673.93   166.6 1671.19     183  1670.3     196 1668.47
   215.7 1668.63   218.9 1668.16   228.7 1665.61   238.5 1664.91   248.3 1665.69
   258.1 1668.79   267.9 1672.69   274.5 1674.78   307.2 1682.91   343.1 1691.05
   349.6 1691.66   356.2  1693.1     366 1694.06   382.3 1696.72   411.7 1704.24
#Mann= 5 ,-1 , 0
       0     .12       0   59.16     .06       0   66.72     .12       0
   228.7    .045       0   248.3     .12       0
Bank Sta=228.7,248.3
XS Rating Curve= 0 ,0
Exp/Cntr=0.3,0.1

Type RM Length L Ch R = 1 ,4401.9  ,304.3,307.6,309.6
XS GIS Cut Line= 2
     2020362.309      181110.962     2020664.392      180881.795
#Sta/Elev= 30
       0 1700.61     6.5    1700    22.9 1695.69    39.2  1692.4    52.3  1690.5
    68.6 1687.65      85 1685.43    98.1 1682.72   111.1 1680.65     134 1675.58
   143.8 1672.63   147.1 1672.05   163.4 1670.82   186.3 1668.21   192.8 1668.15
   202.7 1667.09   212.5 1666.67   215.7 1666.08  217.32  1665.4   222.3 1663.57
   225.5 1663.47   228.8 1663.91  230.91 1665.43   238.6  1670.9   241.9 1672.37
   261.5 1679.38   307.3    1689   320.3 1692.23     353 1703.02   379.2 1710.32
#Mann= 3 ,-1 , 0
       0     .12       0  217.32    .045       0  230.91     .12       0
Bank Sta=217.32,230.91
XS Rating Curve= 0 ,0
Exp/Cntr=0.3,0.1

Type RM Length L Ch R = 1 ,4094.3  ,319.8,321.4,322.4
XS GIS Cut Line= 3
      2020504.91      181349.512     2020834.239      181157.482
     2020886.374      181094.634
#Sta/Elev= 30
       0 1700.06    9.931697.864    29.3 1692.56   52.351688.251    71.7 1684.12
     101 1680.67   130.3 1676.15   146.6 1674.31  164.241673.294   182.5 1672.09
   211.8  1668.4   224.8 1665.76   228.1 1664.25   234.6 1663.17   241.1 1663.59
   244.4 1664.89   245.6 1665.88   250.9 1670.17   254.2 1671.62   260.7 1673.67
   273.7 1676.25   283.5  1680.1   293.2 1684.72   312.8 1696.19   325.8 1701.95
   342.1 1707.89   371.4 1716.75     391 1721.81   430.2 1728.03   462.9 1736.31
#Mann= 6 ,-1 , 0
       0     .06       0    9.93     .12       0   52.35     .06       0
  164.24     .12       0   224.8    .045       0   245.6     .12       0
Bank Sta=224.8,245.6
XS Rating Curve= 0 ,0
Exp/Cntr=0.3,0.1

Type RM Length L Ch R = 1 ,3772.9  ,218,215,211.6
XS GIS Cut Line= 3
     2020610.139      181638.306     2020908.316      181487.264
     2021015.086      181371.379
#Sta/Elev= 30
       0  1717.4     3.3 1716.14   12.541714.017    22.9 1711.77    32.8 1708.62
    42.6 1707.34    68.8 1700.12    91.8 1696.03   170.4 1678.32   180.2 1674.48
   183.5 1673.68   209.7    1670   235.9 1668.45   242.5  1667.5   245.8 1666.83
   252.9 1663.64   258.9 1663.03     272 1663.34   275.3 1664.66   278.5 1666.67
   285.1 1668.96   294.9 1670.78   311.3 1675.23   379.3 1691.16   398.6 1698.79
   421.1 1711.28   427.5 1713.76   453.2 1719.47   466.1 1721.06   491.8 1725.34
#Mann= 4 ,-1 , 0
       0    .016       0   12.54     .12       0   252.9    .045       0
     272     .12       0
Bank Sta=252.9,272
XS Rating Curve= 0 ,0
Exp/Cntr=0.3,0.1

Type RM Length L Ch R = 1 ,3557.9  ,125,126,126.6
XS GIS Cut Line= 2
     2020719.514      181853.149     2021170.034      181530.233
#Sta/Elev= 30
       0 1736.16    65.6 1717.79    68.9 1716.75   73.161713.947    78.7 1709.76
   101.7  1709.1  119.041702.124   167.3  1682.1   177.1 1676.88   203.4 1673.68
   213.2 1665.36   215.8  1664.1     223 1662.72   232.9 1663.96   255.8 1666.46
     269 1666.68   288.6 1669.75   318.2 1671.76     328 1673.18   357.5 1682.24
   370.6 1684.59   380.5 1688.12   406.7 1694.58   419.8 1699.26   446.1 1710.65
   462.5 1715.57   488.7 1716.18   514.9 1720.44   541.2 1722.08   554.3 1723.86
#Mann= 5 ,-1 , 0
       0     .12       0   73.16    .016       0  119.04     .12       0
   215.8    .045       0   232.9     .12       0
Bank Sta=215.8,232.9
XS Rating Curve= 0 ,0
Exp/Cntr=0.3,0.1

Type RM Length L Ch R = 1 ,3431.9  ,369.7,370.1,369
XS GIS Cut Line= 2
     2020801.545       181922.16     2021232.534      181614.868
#Sta/Elev= 30
       0 1723.83   51.421711.361    62.1 1708.93   68.16 1706.16    71.9  1704.3
    75.2 1703.48      85 1703.62    91.5 1702.98   101.3 1700.03  119.041693.089
   156.8 1681.88  169.921680.039   192.8 1678.75   202.6 1677.16   212.4  1674.8
     232 1667.78  256.27 1662.88   264.7 1662.48   273.2 1662.88   300.6 1666.01
   320.2  1670.5   359.4 1683.84     379 1691.58   401.9 1698.18   434.6 1708.82
   444.4 1712.39   457.4 1718.53   473.8 1724.93   506.4  1733.4   529.3 1738.19
#Mann= 7 ,-1 , 0
       0     .12       0   51.42     .06       0   68.16    .016       0
  119.04     .06       0  169.92     .12       0  256.27    .045       0
   273.2     .12       0
Bank Sta=256.27,273.2
XS Rating Curve= 0 ,0
Exp/Cntr=0.3,0.1

Type RM Length L Ch R = 1 ,3061.8  ,255.5,251.2,246.6
XS GIS Cut Line= 2
     2020981.232      182195.597     2021371.857      181935.181
#Sta/Elev= 30
       0 1758.43    29.3 1748.34    61.9 1740.15      75 1735.39      88 1732.06
   110.8 1722.02   123.9  1718.5  130.791715.616   136.9 1710.02   140.2 1709.16
   153.2 1709.43   156.5    1709   159.8 1707.68  173.071695.954   179.3 1689.06
   185.8 1682.78   189.1 1678.67   195.6 1669.06   198.9 1665.39   202.1 1662.06
   205.4 1660.37   221.7 1659.76  229.91 1660.22     238 1662.75   244.5    1664
   264.1 1665.19   361.9 1674.99   391.2 1679.29   456.4 1690.93   469.5 1692.47
#Mann= 5 ,-1 , 0
       0     .12       0  130.79    .016       0  173.07     .12       0
   205.4    .045       0  229.91     .12       0
Bank Sta=205.4,229.91
XS Rating Curve= 0 ,0
Exp/Cntr=0.3,0.1

Type RM Length L Ch R = 1 ,2810.6  ,221.5,218.3,214.4
XS GIS Cut Line= 2
     2021184.345      182393.435     2021515.099      182060.259
#Sta/Elev= 30
       0 1769.07      13 1762.56    42.4  1750.3    68.5 1737.85    81.5 1732.69
    94.6  1725.9   110.8 1720.08   114.71717.554   120.6 1711.53   123.9 1709.46
   136.9 1709.39   140.2 1709.07   143.4 1707.62  156.491694.679     163 1689.66
   172.8 1683.67   208.6 1666.02   221.7 1661.45     238 1657.86   247.8 1656.65
   270.6  1656.1   277.1 1656.71   280.4 1657.88   286.9 1662.33   290.2 1663.72
   299.9 1666.14     326 1668.86   335.8 1668.85   391.2 1675.25   469.5 1689.78
#Mann= 5 ,-1 , 0
       0     .12       0   114.7    .016       0  156.49     .12       0
   247.8    .045       0   277.1     .12       0
Bank Sta=247.8,277.1
XS Rating Curve= 0 ,0
Exp/Cntr=0.3,0.1

Type RM Length L Ch R = 1 ,2592.3  ,177.6,181.1,184.4
XS GIS Cut Line= 3
     2021414.826      182505.493     2021582.795      182268.514
     2021616.649      182092.733
#Sta/Elev= 30
       0 1721.51     3.3    1720   22.161714.604    26.1  1713.2    32.6 1707.32
    35.9 1705.22    45.7  1705.5    55.5 1704.83    58.8 1703.63   64.821698.841
    68.5 1696.17    84.9 1689.71   101.2 1681.68   130.6 1670.82   146.9 1663.66
   156.7 1660.79   169.7  1654.3   175.9  1653.1   182.8 1652.78   195.8 1653.16
   208.9 1654.88   215.4 1656.83   238.2 1657.26   290.5 1660.24   329.5 1665.82
   384.9 1675.19   397.9  1678.9   420.7 1687.06   433.7 1690.75   469.5 1697.56
#Mann= 5 ,-1 , 0
       0     .12       0   22.16    .016       0   64.82     .12       0
   175.9    .045       0   195.8     .12       0
Bank Sta=175.9,195.8
XS Rating Curve= 0 ,0
Exp/Cntr=0.3,0.1

Type RM Length L Ch R = 1 ,2411.2  ,293.9,263,230.7
XS GIS Cut Line= 2
     2021516.389      182618.774     2021867.951      182255.493
#Sta/Elev= 30
       0 1723.11     6.5 1720.85    19.6 1717.88    32.6 1712.92    48.9 1708.02
    68.5 1700.17   72.871697.224    78.3    1694    91.3 1694.15   101.1 1692.93
  114.441685.506   123.9 1681.38   143.5  1674.5   153.3  1669.6   163.1  1666.8
   176.1 1657.45   179.4 1655.93   206.7 1650.79     225 1650.11   231.6 1650.93
   241.4 1654.32   247.9 1655.09   283.8 1652.83   326.2 1652.72   388.1 1649.21
   420.7 1648.64   453.4 1649.06   476.2 1653.23   489.2 1657.59   505.5 1666.54
#Mann= 5 ,-1 , 0
       0     .12       0   72.87    .016       0  114.44     .12       0
   206.7    .045       0   231.6     .12       0
#XS Ineff= 2 , 0
                          247.16         1667.86
Permanent Ineff=
       F       F
Bank Sta=206.7,231.6
XS Rating Curve= 0 ,0
Exp/Cntr=0.3,0.1

Type RM Length L Ch R = 1 ,2148.2  ,353.1,386.3,418.1
XS GIS Cut Line= 4
     2021822.378      182790.649     2021890.086      182613.566
     2021795.034      182474.243     2021934.357      182260.701
#Sta/Elev= 30
       0 1699.44   70.861679.831    78.4 1677.66    88.3 1671.29   107.9 1671.92
   114.4 1670.87  116.97 1669.18   120.9 1666.43     134 1663.83   150.4 1662.79
   160.2 1663.89   192.8  1661.4   196.1 1660.47   199.3 1657.77     209  1646.8
   226.6 1646.31   254.4 1645.19   280.4 1646.85   296.6 1649.26   312.8 1648.28
   338.8 1650.36   361.5 1650.71   430.2 1650.48     453 1648.72   479.2 1649.12
   554.4 1646.59   560.9 1648.04   570.7  1653.6   593.6 1670.64   613.2 1686.74
#Mann= 5 ,-1 , 0
       0     .12       0   70.86    .016       0  116.97     .12       0
     209    .045       0   226.6     .12       0
#XS Ineff= 2 , 0
                          296.31         1657.27
Permanent Ineff=
       F       F
Bank Sta=209,226.6
XS Rating Curve= 0 ,0
Exp/Cntr=0.3,0.1

Type RM Length L Ch R = 1 ,1761.9  ,274.9,298.5,320
XS GIS Cut Line= 2
     2021887.803      182727.181     2022215.287      182402.294
#Sta/Elev= 30
       0 1670.63     9.8  1670.7    13.1  1670.1    22.9 1664.51   30.351661.786
    39.3 1659.36    58.9 1656.23    75.2 1654.64    81.8 1654.78    94.9 1652.53
   114.5 1651.46   153.8 1646.77   199.6 1644.03   242.1    1644   261.7 1642.91
   278.1 1642.96   297.7 1640.08   310.8  1640.9     321 1637.15   330.4 1636.45
     336 1636.63   350.1 1638.24   359.9 1642.32     373 1654.72   382.8 1665.15
   399.1 1678.78   415.5 1690.54   435.1 1703.08   448.2 1709.76   461.3  1715.4
#Mann= 4 ,-1 , 0
       0    .016       0   30.35     .12       0     321    .045       0
     336     .12       0
Bank Sta=321,336
XS Rating Curve= 0 ,0
Exp/Cntr=0.3,0.1

Type RM Length L Ch R = 1 ,1463.4  ,209,193.7,177.7
XS GIS Cut Line= 4
     2021912.222      182814.087     2022088.003      182719.035
     2022250.764      182754.191     2022396.597      182695.597
#Sta/Elev= 30
       0 1680.18   12.631676.228    16.4 1673.25    19.7 1669.33    39.3 1669.11
    42.6  1668.3    49.41664.092    55.7  1660.9    68.8 1657.05    88.4 1652.08
   111.4  1647.6   137.6 1645.49   147.4 1643.54   183.4 1642.03   199.8 1638.93
   209.6 1639.16   252.1 1636.12   284.7 1630.82   297.8 1632.88   310.8 1631.98
   336.2 1632.17   340.2 1632.59   353.3 1638.56   369.6 1640.51   382.7 1644.01
   402.4 1647.58   454.8 1661.42   484.2 1667.76   500.6 1673.58   523.5 1683.57
#Mann= 5 ,-1 , 0
       0     .12       0   12.63    .016       0    49.4     .12       0
   310.8    .045       0   336.2     .12       0
Bank Sta=310.8,336.2
XS Rating Curve= 0 ,0
Exp/Cntr=0.3,0.1

Type RM Length L Ch R = 1 ,1269.7  ,160.2,154,146.6
XS GIS Cut Line= 3
     2022011.253      183018.673     2022282.954      182878.916
     2022341.982      182796.451
#Sta/Elev= 30
       0 1672.71     6.5 1671.68     9.8 1670.23    16.2 1664.88    19.5 1663.76
    29.2 1664.57    35.8 1664.06      39 1662.84    48.8 1655.08    61.8 1646.08
    74.8 1636.35      91 1631.66     104 1630.38     130 1629.58     156 1630.51
   162.5 1631.33   165.8 1630.68   175.5 1626.87   183.5 1625.55   191.8 1624.89
   198.5  1625.3     208 1626.48   214.5 1628.21   224.3 1629.74   243.8 1631.06
   276.3 1637.64   348.1 1645.08   361.2 1647.26   377.5 1651.35     407 1656.83
#Mann= 5 ,-1 , 0
       0     .12       0    19.5    .016       0    61.8     .12       0
   183.5    .045       0   198.5     .12       0
Bank Sta=183.5,198.5
XS Rating Curve= 0 ,0
Exp/Cntr=0.3,0.1

Type RM Length L Ch R = 1 ,1115.7  ,222.6,226.8,231.2
XS GIS Cut Line= 4
     2022103.266      183151.486     2022187.468      183106.347
     2022308.996      182987.423     2022368.023       182881.52
#Sta/Elev= 30
       0 1663.73    15.9 1659.66    38.2 1656.25    44.6 1653.74    47.8 1650.59
      51 1648.99    73.2 1648.08    89.2 1643.45    98.8 1638.91   102.1 1636.45
   111.9 1624.73  114.03 1623.69   121.7 1622.68   125.4 1622.82   140.4 1622.89
   157.7 1623.11   170.8 1625.75   180.6 1626.57   206.7 1626.81     246 1625.61
   249.2 1626.26   265.6  1634.5   275.4 1636.15     282  1635.7   298.3 1630.97
   308.2 1631.17   334.4 1635.67   344.2 1639.22     354 1640.94   386.8 1649.71
#Mann= 5 ,-1 , 0
       0     .12       0    44.6    .016       0    89.2     .12       0
   125.4    .045       0   140.4     .12       0
Bank Sta=114.03,140.4
XS Rating Curve= 0 ,0
Exp/Cntr=0.3,0.1

Type RM Length L Ch R = 1 ,888.9   ,315.7,312.4,306.6
XS GIS Cut Line= 4
     2022215.607      183295.424     2022309.357      183269.382
     2022508.576      183127.889     2022551.545      183066.691
#Sta/Elev= 30
       0 1656.65    19.5 1654.48    87.6 1640.57   103.8 1637.57   113.6 1636.56
  115.141635.583   120.1 1632.21   123.4 1631.53   136.4 1632.33  148.021631.417
   162.5 1626.63     169    1622   172.2 1621.22   191.8 1620.82   200.2 1618.96
   208.1 1618.06   217.8  1618.9   224.4 1620.01   279.8 1619.55   302.6 1617.75
   312.3 1618.92   315.6 1620.01   331.9 1629.53   344.9 1639.06   351.4 1644.43
   370.9 1656.84   380.7 1662.44   390.4 1669.49   406.7 1680.22   416.4 1688.96
#Mann= 5 ,-1 , 0
       0     .12       0  115.14    .016       0  148.02     .12       0
   200.2    .045       0   217.8     .12       0
Bank Sta=200.2,217.8
XS Rating Curve= 0 ,0
Exp/Cntr=0.3,0.1

Type RM Length L Ch R = 1 ,576.5   ,497.3,495.8,494.5
XS GIS Cut Line= 3
     2022361.441       183524.59     2022475.044      183496.292
     2022707.795      183280.233
#Sta/Elev= 30
       0  1650.1     9.8 1647.99   100.8 1632.58  112.881631.212   117.1 1630.53
   123.6  1626.3   143.3 1625.96   146.5 1624.42   149.8 1621.59   156.4 1614.03
   159.6 1612.62   166.2    1612   178.2 1612.76  178.341612.777   195.6 1614.36
   208.8 1613.24   231.7 1613.09  235.861613.924   244.8 1615.84   251.3 1616.46
   274.2 1616.67   303.7 1618.01   320.1 1617.96   333.2  1619.7   346.2 1623.19
   382.3 1635.86   401.9 1644.12   411.7 1647.42   424.8 1653.74   434.6 1657.73
#Mann= 6 ,-1 , 0
       0     .12       0  112.88    .016       0   159.6    .045       0
   178.2     .12       0  178.34    .016       0  235.86     .12       0
Bank Sta=159.6,178.2
XS Rating Curve= 0 ,0
Exp/Cntr=0.3,0.1
